--- dmsfrk.prj (project) ---

Proj Title=dmsfrk
Current Plan=p01
Default Exp/Contr=0,0
English Units
Geom File=g01
Flow File=f01
Plan File=p01
BEGIN DESCRIPTION:
END DESCRIPTION:
DSS Export Rating Curves= 0
DSS Export Rating Curve Sorted= 0
DSS Export Volume Flow Curves= 0
DXF OffsetX= 0
DXF OffsetY= 0
DXF ScaleX= 0
DXF ScaleY= 0

--- dmsfrk.p01 (plan) ---

Plan Title=Floodplain
Program Version=4.00
Geom File=g01
Flow File=f01
K Sum by GR=0
Std Step Tol=0.01
Critical Tol=0.01
Num of Std Step Trials=20
Max Error Tol=0.3
Flow Tol Ratio=0.001
Split Flow NTrial=30
Split Flow Tol=0.02
Split Flow Ratio=0.02
Log Output Level=0
Friction Slope Method=1
Unsteady Friction Slope Method=2
Unsteady Bridges Friction Slope Method=1
Global Log Level=0
CheckData=False
Run HTab=0
Run UNet=0
Run PostProcess=0
UNET Theta=0
UNET Theta Warmup=0
UNET ZTol=0
UNET ZSATol=0
UNET MxIter=0
UNET MaxInSteps=0
UNET DtIC=0
UNET DtMin=0
UNET MaxCRTS=0
UNET WFStab=0
UNET SFStab=0
UNET WFX=0
UNET SFX=0
UNET DSS MLevel=0
UNET DZMax Abort=0
UNET Convert EG Bridges=0
UNET Use Existing IB Tables=0
UNET Froude Limit=0
UNET Froude Power=0
Write IC File=0
Echo Input=False
Echo Output=False
Write Detailed=0

--- dmsfrk.f01 (steady flow) ---

Flow Title=NFF Regression Equation
Program Version=4.00
Number of Profiles=1
Profile Names=P100yr
River Rch & RM=dmsfrk,Main      ,33775.8
     355
River Rch & RM=dmsfrk,Main      ,33556.4
     355
River Rch & RM=dmsfrk,Main      ,33373
     442
River Rch & RM=dmsfrk,Main      ,32460.2
     474
River Rch & RM=dmsfrk,Main      ,30937
     512
River Rch & RM=dmsfrk,Main      ,28867
     566
River Rch & RM=dmsfrk,Main      ,28288.8
     613
River Rch & RM=dmsfrk,Main      ,25757.4
     672
River Rch & RM=dmsfrk,Main      ,24710.3
     744
River Rch & RM=dmsfrk,Main      ,23195
     767
River Rch & RM=dmsfrk,Main      ,21622.3
     850
River Rch & RM=dmsfrk,Main      ,21166.9
    1374
River Rch & RM=dmsfrk,Main      ,20994.5
    1534
River Rch & RM=dmsfrk,Main      ,16282.2
    1667
River Rch & RM=dmsfrk,Main      ,15948.9
    1960
River Rch & RM=dmsfrk,Main      ,15016.4
    1969
River Rch & RM=dmsfrk,Main      ,9216.1
    2187
Boundary for River Rch & Prof#=dmsfrk,Main      ,1
Up Type=0
Dn Type=3
Dn Slope=0.010512

--- dmsfrk.g01 (geometry) ---

Geom Title=USGS 10m DEM
Program Version=4.00

River Reach=dmsfrk          ,Main
Reach XY= 30
     1649943.792      263226.405     1648910.202       263482.22
     1647678.385        264203.3     1646732.211      263730.117
     1645430.086      263637.238     1642495.266       265137.21
     1641566.731      266946.151     1640283.406      268054.637
     1639657.685      267961.092     1638861.041      269046.518
     1638237.624      268987.222      1638120.15      269666.456
     1637271.177      270080.978     1636397.236      270233.078
      1635257.38       269580.82       1633921.3      269298.865
      1633379.88      269724.037      1632824.36      269090.185
     1632632.375      269404.409     1632836.057      269927.157
     1631944.345      270240.912     1630805.775      271108.222
     1630249.799       270713.66     1629341.834      270739.214
     1628369.187      269891.142     1627382.165      269784.135
     1626991.987       269280.52     1625404.138       269132.35
     1624955.398      268667.882     1624296.354      269632.109

Type RM Length L Ch R = 1 ,33775.8 ,209.6,219.4,229.2
XS GIS Cut Line= 4
     1649779.459      262886.134     1649867.547      263145.679
     1649977.657      263291.968     1650314.278      263439.829
#Sta/Elev= 30
     9.8 1336.05    39.2 1315.92    48.9 1314.75    58.7 1308.64   156.6 1220.79
   166.4 1218.84   205.6  1187.7   244.7 1161.98   264.3 1150.55   274.1 1149.88
   331.9 1125.93   341.5    1124   360.5 1123.27   370.5 1123.09   380.5 1123.35
   389.7 1124.39   428.3 1133.43   477.1 1150.19     487 1155.67   496.9 1163.58
   546.6 1189.41   576.4 1202.27   655.9 1246.04   675.8 1261.35   705.6 1274.43
   745.4 1303.06   765.2 1321.66   785.1  1333.5     805 1342.61   824.8 1347.49
#Mann= 3 , 0 , 0
       0      .1       0   360.5    .045       0   380.5      .1       0
Bank Sta=360.5,380.5
XS Rating Curve= 0 ,0
Exp/Cntr=0.3,0.1

Type RM Length L Ch R = 1 ,33556.4 ,175.8,183.4,190.9
XS GIS Cut Line= 4
     1649608.002      263016.693     1649747.999      263287.249
     1649788.897      263439.829     1649751.145      263756.002
#Sta/Elev= 30
     9.8 1284.35   108.1  1223.1   127.7 1216.28   157.2 1199.68   176.9 1189.79
   196.5 1181.28     226 1165.86   235.8 1161.72   275.1 1153.22   304.6  1140.6
     354 1123.32   373.6 1120.45   383.6 1119.22   393.6 1119.46   413.2 1120.63
   462.6 1137.57   472.5 1137.93   482.5 1140.92   522.3 1159.22   542.2 1170.13
   562.1 1182.34   572.1 1184.62     582 1188.23   601.9 1199.02   621.8 1208.43
   661.6  1225.1   681.5  1229.4   761.1 1271.03   771.1 1275.59     781 1275.91
#Mann= 3 , 0 , 0
       0      .1       0   373.6    .045       0   393.6      .1       0
Bank Sta=373.6,393.6
XS Rating Curve= 0 ,0
Exp/Cntr=0.3,0.1

Type RM Length L Ch R = 1 ,33373   ,169.7,166.7,163.6
XS GIS Cut Line= 4
     1649571.823      262997.817     1649596.991      263299.833
     1649590.699      263455.559      1649727.55      263767.013
#Sta/Elev= 30
    10.1 1297.96    20.2 1296.19    50.5 1278.53     101 1254.76   111.1 1250.59
   121.2 1249.45   212.1 1204.44   222.2 1200.07   232.3 1199.38   252.6 1190.76
   262.7  1185.1   322.5 1140.26   332.3 1140.14   361.5 1118.21     371 1113.89
     381  1113.1     391 1114.73     420 1122.73   458.9 1125.25   468.9    1128
   488.9 1138.17     529 1160.19     559 1170.76     589 1186.74     649 1215.16
     669 1220.24   739.1 1261.39   749.1  1266.1   769.1 1272.94   799.1 1277.14
#Mann= 3 , 0 , 0
       0      .1       0     371    .045       0     391      .1       0
Bank Sta=371,391
XS Rating Curve= 0 ,0
Exp/Cntr=0.3,0.1

Type RM Length L Ch R = 1 ,33206.4 ,180,183.1,186.1
XS GIS Cut Line= 4
     1649431.468      263084.854      1649421.53      263309.161
     1649435.727       263479.52     1649363.324      263747.837
#Sta/Elev= 30
     9.8 1264.86    19.5  1263.8    48.8 1250.93    78.1 1241.09    87.9 1236.67
   107.4 1224.01   126.9 1217.49     166  1192.8   214.8 1157.31   224.5  1157.3
   274.8 1118.32   284.9 1111.26     295 1107.69     305 1107.15     315 1108.68
   325.1 1108.95   395.5  1136.7   415.3 1143.24   425.3 1143.93   435.2 1146.48
     455 1158.08   474.9 1167.91   524.5 1188.58   534.4 1188.81   554.3 1197.98
   623.8  1239.2   643.6 1245.21   653.5  1249.7   663.5 1252.76   673.4 1254.05
#Mann= 3 , 0 , 0
       0      .1       0     295    .045       0     315      .1       0
Bank Sta=295,315
XS Rating Curve= 0 ,0
Exp/Cntr=0.3,0.1

Type RM Length L Ch R = 1 ,33023.3 ,88.8,89.5,90.2
XS GIS Cut Line= 4
     1649302.841      263041.861     1649254.078      263321.855
     1649247.786      263476.008     1649277.673      263756.002
#Sta/Elev= 30
     9.8 1305.05    29.4 1291.91    39.2 1288.13      49 1285.33   117.6 1237.17
   137.2 1224.33     147 1223.82   205.8  1189.5   235.2 1170.95     245 1167.38
   254.8 1164.78   284.2 1146.77   342.1  1113.4   351.7 1113.09   370.6 1103.87
   380.6 1102.23   390.6 1102.68   419.2 1111.41   458.6 1120.07   498.8 1142.11
   549.1 1174.16   559.2 1179.28   569.2 1181.72   579.3 1189.74   589.3 1196.27
   609.5 1203.42   649.7 1223.92   659.7 1227.97   669.8 1228.52   720.1 1250.71
#Mann= 3 , 0 , 0
       0      .1       0   370.6    .045       0   390.6      .1       0
Bank Sta=370.6,390.6
XS Rating Curve= 0 ,0
Exp/Cntr=0.3,0.1

Type RM Length L Ch R = 1 ,32933.8 ,90.3,85.5,80.7
XS GIS Cut Line= 4
     1649199.023      263040.288     1649169.136      263304.552
     1649156.552      263496.457     1649178.574      263748.137
#Sta/Elev= 30
     9.8 1315.27    19.7  1307.5    29.5 1302.17    39.4 1298.95    98.5 1244.74
   108.3  1236.5     128 1222.65   137.9 1222.65   167.4 1204.95   226.5 1174.33
   236.4 1172.51   246.2 1168.94   326.7 1120.24   346.9 1113.49   367.3 1099.17
   377.3 1097.76   387.3 1100.73   407.7 1109.39   417.8 1111.27   458.3 1114.29
   468.4 1117.01   478.5 1121.25   539.1 1152.19   559.3 1158.23   579.5    1172
     620 1202.28   640.2 1214.16   650.3 1217.28   660.4 1218.88   710.9 1244.97
#Mann= 3 , 0 , 0
       0      .1       0   367.3    .045       0   387.3      .1       0
Bank Sta=367.3,387.3
XS Rating Curve= 0 ,0
Exp/Cntr=0.3,0.1

Type RM Length L Ch R = 1 ,32848.3 ,235.6,225.9,216.3
XS GIS Cut Line= 4
     1649159.698      263057.591     1649063.745      263307.698
      1649087.34      263493.311     1649153.406      263738.699
#Sta/Elev= 30
     9.9 1297.33    19.8 1297.19    59.5  1270.7   109.1 1236.08     129 1229.53
   168.7 1199.44   198.4 1179.34   208.4 1173.69   218.3 1170.57   228.2 1169.75
     248 1162.97   287.6 1139.16   317.1  1119.1     327 1116.77   336.8 1113.05
   346.7 1107.78   376.1 1095.61   386.1 1094.21   396.1 1096.41   415.6 1105.63
   425.4 1107.21   445.1 1108.25     455 1111.36   533.2 1152.56   552.7 1157.28
   572.3 1168.37   650.5 1215.95   660.2 1217.44     670 1220.77   709.1 1236.24
#Mann= 3 , 0 , 0
       0      .1       0   376.1    .045       0   396.1      .1       0
Bank Sta=376.1,396.1
XS Rating Curve= 0 ,0
Exp/Cntr=0.3,0.1

Type RM Length L Ch R = 1 ,32622.4 ,160.7,162.2,163.8
XS GIS Cut Line= 4
      1648541.51      263244.778     1648845.099      263463.424
     1648897.008      263556.231     1648972.511      263807.911
#Sta/Elev= 30
    10.1 1247.41    50.6 1219.88    60.7 1207.64    70.8 1197.94      91 1182.64
   121.3 1162.98   151.7 1147.99   161.8  1139.2     182 1129.71   202.2 1122.53
   232.6 1113.59   262.9 1108.49   333.7 1107.69     364 1108.52   393.5 1105.28
   403.1 1101.72   422.1 1089.42   432.1 1088.07   442.1 1090.86   461.1 1097.51
   480.5 1106.87   490.6 1110.39     531 1143.53   551.2 1156.58   581.5 1177.86
   591.6 1179.16   642.2 1209.96   682.6 1233.31   692.7 1238.24   743.2 1250.08
#Mann= 3 , 0 , 0
       0      .1       0   422.1    .045       0   442.1      .1       0
Bank Sta=422.1,442.1
XS Rating Curve= 0 ,0
Exp/Cntr=0.3,0.1

Type RM Length L Ch R = 1 ,32460.2 ,247.5,243.5,239.4
XS GIS Cut Line= 4
     1648428.254      263326.574     1648703.529      263532.636
     1648760.157      263650.611      1648871.84      263858.247
#Sta/Elev= 30
    10.1 1279.99    20.2  1272.4   101.1 1228.72   121.4 1211.88   131.5 1205.87
   141.6 1200.06   161.8 1190.82   202.3  1168.8   222.5 1154.15   232.6 1149.21
   262.9 1135.04   303.4 1118.57   323.6 1109.23   343.9 1103.61   353.9 1102.79
   374.1 1097.99   384.1 1096.66   394.2  1093.8   404.3 1088.69   414.3 1085.64
   424.3 1086.98   454.6 1102.33   464.7 1104.01   484.5 1114.46     514 1137.09
   582.8    1183   592.6 1184.66   651.5 1221.67   690.8  1244.8   710.5  1251.2
#Mann= 3 , 0 , 0
       0      .1       0   404.3    .045       0   424.3      .1       0
Bank Sta=404.3,424.3
XS Rating Curve= 0 ,0
Exp/Cntr=0.3,0.1

Type RM Length L Ch R = 1 ,32216.7 ,410.2,408.8,407.4
XS GIS Cut Line= 4
     1648237.922      263534.209     1648485.796      263665.124
     1648578.267      263798.052     1648716.113      263977.794
#Sta/Elev= 30
      10 1263.82    80.1 1226.99    90.1 1219.63   120.1 1202.64   130.1 1198.56
   150.2 1193.69   170.2 1182.36   190.2 1168.39   250.3 1131.19   260.3 1124.11
   280.3 1106.66   300.6 1091.01   310.7 1087.01   320.8 1087.58   330.9 1086.56
     341 1082.07   351.3 1081.29   361.3  1080.3   371.3 1082.85   391.6 1094.64
     422 1116.42   461.9 1140.75   481.6 1149.39   491.5 1151.58   550.6 1179.85
   570.3 1192.51   619.5 1217.84   629.4 1219.78   639.2 1224.68   668.8 1242.21
#Mann= 3 , 0 , 0
       0      .1       0   351.3    .045       0   371.3      .1       0
Bank Sta=351.3,371.3
XS Rating Curve= 0 ,0
Exp/Cntr=0.3,0.1

Type RM Length L Ch R = 1 ,31807.9 ,357.9,375.9,393.9
XS GIS Cut Line= 4
     1648017.702      263680.498     1648126.239      263872.404
     1648233.203      264009.254     1648458.141      264160.262
#Sta/Elev= 30
      10  1285.1      20 1277.16    40.1 1257.79    90.2 1215.93   110.2 1202.36
   120.3 1197.27   200.4  1135.1   220.5 1117.81   230.1 1113.06   239.8 1110.92
     288 1080.43   297.7 1076.81     307  1075.2     317  1073.9     327 1074.23
   336.3 1075.73   365.2 1088.56   384.5 1096.09   394.2 1098.55   434.3 1114.57
   444.3 1118.97   464.4 1130.63   544.7 1166.89   564.7 1179.41   574.8 1183.65
   584.8 1185.68   594.9 1190.88   614.9 1197.08     645 1210.14   665.1 1221.36
#Mann= 3 , 0 , 0
       0      .1       0     307    .045       0     327      .1       0
Bank Sta=307,327
XS Rating Curve= 0 ,0
Exp/Cntr=0.3,0.1

Type RM Length L Ch R = 1 ,31432   ,248.1,244.4,239.7
XS GIS Cut Line= 4
     1647854.111      263817.349      1647885.57      264006.108
     1647874.559      264196.441       1647901.3      264473.289
#Sta/Elev= 30
    10.1 1239.08    30.2 1224.96    40.3 1224.55    60.4 1210.64    70.5 1202.01
    80.6 1192.18   110.8 1158.24     141 1130.69   151.1 1128.97   181.3 1107.38
   191.4 1101.02   221.5 1085.92   241.5 1079.24   251.6 1078.24   291.7 1069.25
   301.7  1068.3   311.7  1068.7   361.9 1074.62     382  1082.1   441.6 1107.41
   451.5 1110.11   461.5 1111.63   481.3 1120.17   501.2 1125.61   511.1 1130.53
   560.8 1159.88   570.7 1160.35   630.3 1197.02   640.3  1202.2   660.2  1209.8
#Mann= 3 , 0 , 0
       0      .1       0   291.7    .045       0   311.7      .1       0
Bank Sta=291.7,311.7
XS Rating Curve= 0 ,0
Exp/Cntr=0.3,0.1

Type RM Length L Ch R = 1 ,31187.6 ,220,250.6,281.6
XS GIS Cut Line= 4
     1647760.523      263858.571     1647665.405      264145.343
      1647685.28      264248.978     1647696.638      264467.607
#Sta/Elev= 30
    10.1 1201.63    30.2 1186.42    60.4 1159.24    80.6 1143.26    90.6 1140.34
   100.7 1134.73   130.9  1111.4   151.1 1097.34   181.3 1078.66   191.4 1073.56
   201.4 1073.03   211.5  1070.4   271.9 1070.98   321.3 1070.07   330.9 1069.39
   349.7 1064.43   359.7 1062.76   369.7 1065.77   388.5 1086.23   398.1 1094.35
   407.7 1096.12   447.5 1113.37   477.3 1124.81   497.2 1134.19   517.1 1139.17
     537 1148.62   576.8 1165.18   606.7 1179.65   616.6  1183.1   626.6 1184.45
#Mann= 3 , 0 , 0
       0     .08       0   349.7    .045       0   369.7     .08       0
Bank Sta=349.7,369.7
XS Rating Curve= 0 ,0
Exp/Cntr=0.3,0.1

Type RM Length L Ch R = 1 ,30937   ,235.8,218.2,201.3
XS GIS Cut Line= 4
     1647758.158      263829.933     1647616.588      263991.951
     1647446.704      264086.331     1647212.328      264355.314
#Sta/Elev= 30
     9.8 1213.61    19.6 1209.38    58.7 1180.49   117.4 1134.26   127.1  1124.5
   146.7 1115.58     176 1097.41   205.4 1081.55   224.9 1072.65   234.6 1069.57
   263.7  1068.2   292.9 1064.96   321.8 1057.75   331.8  1057.7   341.8 1058.58
   419.4 1068.21   429.3 1071.68   439.2 1077.06     459 1082.04   478.9 1092.63
   488.8  1095.9   508.6 1100.48   558.1 1114.51   568.1 1116.76     578  1117.6
   617.6 1133.51     687 1168.72   696.9 1175.77   736.5 1190.53   766.3 1197.33
#Mann= 3 , 0 , 0
       0     .08       0   321.8    .045       0   341.8     .08       0
Bank Sta=321.8,341.8
XS Rating Curve= 0 ,0
Exp/Cntr=0.3,0.1

Type RM Length L Ch R = 1 ,30718.8 ,264.1,239,213.9
XS GIS Cut Line= 4
     1647522.208      263675.779     1647363.335      263873.976
     1647306.707      264021.838     1647198.171      264334.865
#Sta/Elev= 30
     9.8 1209.88    39.1 1180.37    48.8 1178.43    87.9 1155.98   156.3 1123.22
   166.1 1119.64   175.9 1119.25   214.9 1107.98   234.5 1106.09   244.2 1102.22
     254 1094.84   273.8 1076.71   293.6 1066.23   303.5 1057.46  308.01 1055.88
   313.4 1054.21   333.2 1055.63   432.4 1064.35   452.5 1068.87   492.7 1088.12
   502.7 1089.44   512.7 1092.95     573 1120.96     583 1126.33   593.1 1133.57
   603.1 1135.75   663.3    1175   673.4  1180.2   693.5 1187.48   743.7 1196.28
#Mann= 3 , 0 , 0
     9.8     .08       0  308.01    .045       0   333.2     .08       0
Bank Sta=308.01,333.2
XS Rating Curve= 0 ,0
Exp/Cntr=0.3,0.1

Type RM Length L Ch R = 1 ,30479.8 ,135.3,168.5,201.8
XS GIS Cut Line= 4
     1647106.937      263527.917     1647080.196      263847.236
     1647161.992      263962.064     1647177.722       264311.27
#Sta/Elev= 30
      10 1153.06      30 1138.55    80.1  1121.9   130.2 1113.03   190.3 1107.59
   220.3 1100.81   240.3 1094.73   250.3 1093.84   300.4 1074.76   340.6 1067.53
   350.6 1064.09   370.8 1052.89   380.9 1049.27   390.9 1049.25   400.9 1050.22
   501.4 1056.19   511.4 1057.41   521.3 1060.61   571.3  1086.3   581.3 1090.42
   591.3 1091.47   641.2 1117.06   651.2 1122.29   671.2 1138.29   691.1 1151.68
   701.1  1151.8   731.1  1170.3     761 1185.64     781 1192.56     811 1195.29
#Mann= 3 , 0 , 0
       0     .06       0   380.9    .045       0   400.9     .06       0
Bank Sta=380.9,400.9
XS Rating Curve= 0 ,0
Exp/Cntr=0.3,0.1

Type RM Length L Ch R = 1 ,30311.2 ,238.2,235.3,232.5
XS GIS Cut Line= 4
     1647091.207      263531.063     1647062.893      263831.506
     1646916.604      264007.681     1646839.527      264160.262
#Sta/Elev= 30
    10.1 1153.43    30.2  1138.1    40.2 1137.02    60.4 1127.13    70.4 1123.71
   120.7    1114     171 1109.29   201.2 1103.82   231.4 1093.15   251.5  1088.8
   281.7 1075.63   301.8  1070.5   381.4 1066.34   391.4 1064.52   401.3 1060.34
   421.2 1048.63   431.2 1044.57   441.2 1043.29   451.2 1043.99     481 1045.74
   490.9 1048.27   510.9 1066.69   540.8 1091.41   550.9 1096.92   591.1 1109.29
   611.2 1124.57   631.3 1136.01   641.4 1143.41   691.7 1185.18   701.7 1186.47
#Mann= 3 , 0 , 0
       0     .06       0   431.2    .045       0   451.2     .06       0
Bank Sta=431.2,451.2
XS Rating Curve= 0 ,0
Exp/Cntr=0.3,0.1

Type RM Length L Ch R = 1 ,30075.9 ,310.2,286.3,262.4
XS GIS Cut Line= 4
      1646951.21      263491.738     1646850.538      263704.093
     1646746.721      263861.393     1646707.396       264106.78
#Sta/Elev= 30
     9.8  1175.7      49 1150.55    58.8 1145.54    68.5 1143.75   107.7 1119.08
   137.1 1103.09   166.5 1089.11   176.3 1087.85   254.8 1052.93   274.7  1048.7
   294.5 1047.38   324.2 1038.39   334.2 1038.02   344.2 1038.43   383.8 1041.12
   393.7 1045.52   403.6 1046.63   423.5 1059.75   463.2    1090   473.2 1095.58
   483.1 1098.79   512.9 1103.08   522.9 1108.06   562.7 1131.26   602.4 1158.42
   612.4 1159.89   642.2 1184.73   652.1 1191.69   662.1 1197.41     672 1201.47
#Mann= 3 , 0 , 0
       0     .06       0   324.2    .045       0   344.2     .06       0
Bank Sta=324.2,344.2
XS Rating Curve= 0 ,0
Exp/Cntr=0.3,0.1

Type RM Length L Ch R = 1 ,29789.6 ,317.5,330.2,343
XS GIS Cut Line= 4
     1646369.201      263409.942     1646506.052      263678.925
     1646570.545      263851.955     1646589.421      264083.185
#Sta/Elev= 30
    10.1 1135.12    40.2 1120.45    70.4 1108.67    80.5 1105.09    90.5 1104.58
   130.8 1091.67   150.9  1087.2   201.2 1079.65   221.3 1077.41   251.5 1069.04
   321.2 1045.22     331 1042.48   340.7 1042.81   350.4  1039.4   360.1 1037.34
   408.4 1034.22   418.4 1033.09   428.4 1033.54   437.9 1036.27   447.6 1036.74
     467 1049.72   496.5 1067.23   526.8 1087.72     547 1099.54   567.1 1104.62
   587.3 1114.67   647.8 1147.92     668 1153.83   688.2 1165.83   718.5 1180.29
#Mann= 3 , 0 , 0
       0     .06       0   408.4    .045       0   428.4     .06       0
Bank Sta=408.4,428.4
XS Rating Curve= 0 ,0
Exp/Cntr=0.3,0.1

Type RM Length L Ch R = 1 ,29459.4 ,241.4,239.3,237.3
XS GIS Cut Line= 4
     1646221.339      263453.986     1646237.069       263702.52
     1646215.047      263847.236     1646260.664      264100.488
#Sta/Elev= 30
      10 1148.53    19.9 1146.91    69.7 1116.35    99.6 1099.09   109.6 1094.06
   119.5 1093.73   139.5 1083.09   179.3 1059.86   219.1 1038.14   229.1 1037.38
   239.1 1035.19     249 1034.13   278.3  1031.8   326.9 1029.19   327.1 1029.18
   336.9 1029.18   346.9 1030.19   356.4 1034.18   366.1  1041.9   375.9 1048.78
   425.1 1078.13     435 1078.34   454.8 1089.47   484.5  1107.5   524.1 1129.71
   543.9 1135.11   603.3  1169.9   632.9 1188.65   642.8 1194.46   652.7 1194.89
#Mann= 3 , 0 , 0
       0     .06       0   326.9    .045       0   346.9     .06       0
Bank Sta=326.9,346.9
XS Rating Curve= 0 ,0
Exp/Cntr=0.3,0.1

Type RM Length L Ch R = 1 ,29220   ,342.7,353,363.3
XS GIS Cut Line= 4
     1646021.569      263464.997     1645993.255      263680.498
     1645980.671       263859.82     1646031.007      264131.948
#Sta/Elev= 30
     9.9 1143.21      79 1105.57    88.9 1105.18   118.6 1088.58   177.8 1053.36
   187.7 1051.73   197.6 1047.47   207.5 1041.45   217.4 1036.95   227.3    1035
   277.3 1029.89   297.2 1028.71  330.78 1024.67   347.2 1023.62  350.13 1024.45
   357.2 1026.59   377.1 1040.96   387.1 1045.08   397.1 1047.06   426.8 1064.76
   466.3 1091.83   476.2 1098.26   486.1 1103.78     496 1108.04   505.8 1108.56
   515.7  1112.4   594.8 1157.63   614.6 1163.43   644.2 1181.29   673.9 1197.78
#Mann= 3 , 0 , 0
     9.9     .06       0  330.78    .045       0  350.13     .06       0
Bank Sta=330.78,350.13
XS Rating Curve= 0 ,0
Exp/Cntr=0.3,0.1

Type RM Length L Ch R = 1 ,28867   ,278,262.4,246.8
XS GIS Cut Line= 4
     1645747.867      263436.683     1645692.812      263666.341
     1645626.746      263793.754     1645510.345      264139.813
#Sta/Elev= 30
     9.8 1146.78    68.9 1105.45    78.7 1099.47    88.6 1098.67   118.1 1079.52
   177.1 1045.89   196.8 1040.32   226.3 1024.06   236.2 1021.77   245.7 1021.12
   312.7  1019.2   331.4 1017.75   341.4 1017.61   351.4 1019.37   370.1 1024.94
   419.2 1029.47   438.9 1031.85   448.8  1034.2   458.6  1039.7   488.2 1061.73
   498.1 1067.51     508 1068.62   557.3  1085.4     577  1091.2   606.6 1098.73
   616.5 1099.38   665.9 1113.83   715.2 1135.24   725.1 1137.84   744.8 1149.59
#Mann= 3 , 0 , 0
       0     .06       0   331.4    .045       0   351.4     .06       0
Bank Sta=331.4,351.4
XS Rating Curve= 0 ,0
Exp/Cntr=0.3,0.1

Type RM Length L Ch R = 1 ,28604.6 ,188.6,177.3,166.1
XS GIS Cut Line= 4
     1645447.425      263398.931     1645445.852       263592.41
     1645460.009      263716.677     1645489.896      264119.364
#Sta/Elev= 30
     9.7 1142.89    19.3 1137.48    38.7 1129.18    77.4 1114.18    96.7 1110.24
   106.4 1104.97   125.8  1091.1   183.8 1043.63   193.5 1043.47   203.1  1036.7
   212.7 1028.32   222.3 1018.97   231.6 1013.47   241.6 1012.69   251.6 1013.83
     369  1020.6   399.3 1023.86   409.4  1024.1   439.7 1028.78   449.8 1031.15
     470 1038.53   500.3 1052.59   510.4 1053.03   601.2 1098.13   611.3 1098.25
   641.6  1113.5   651.7 1117.47     682 1127.26   712.3 1138.24   722.4 1139.66
#Mann= 3 , 0 , 0
       0     .08       0   231.6    .045       0   251.6     .06       0
Bank Sta=231.6,251.6
XS Rating Curve= 0 ,0
Exp/Cntr=0.3,0.1

Type RM Length L Ch R = 1 ,28427.3 ,145.9,138.5,131.1
XS GIS Cut Line= 4
     1645398.662      263431.964     1645260.238      263660.049
     1645340.461      263787.462     1645461.582      264105.207
#Sta/Elev= 30
     9.9 1121.74    19.8  1118.1    39.5  1109.4    49.4 1106.85    59.3 1105.74
   118.6  1088.2   158.1 1070.55     168 1067.97   177.9 1067.39   217.4  1049.5
   237.2  1041.9   266.8 1032.64   286.9 1029.45     307  1020.4   327.1 1009.15
   337.1 1006.87   347.1 1007.89   357.1  1010.8   367.2 1012.82   507.4 1024.15
   537.4 1028.98   567.4 1043.93   637.4 1080.59   647.4 1084.48   657.4 1086.78
   697.4 1109.71   707.4 1113.23   727.4 1123.71   747.4 1132.99   757.4 1135.11
#Mann= 3 , 0 , 0
       0     .08       0   327.1    .045       0   347.1     .06       0
Bank Sta=327.1,347.1
XS Rating Curve= 0 ,0
Exp/Cntr=0.3,0.1

Type RM Length L Ch R = 1 ,28288.8 ,285.5,306.5,327.6
XS GIS Cut Line= 4
     1644947.212      263584.545      1645124.96       263749.71
     1645255.519      263862.966     1645412.819      264120.937
#Sta/Elev= 30
    10.1 1102.23    40.4 1089.23    70.8 1078.32    80.9  1076.6      91 1072.81
   101.1 1071.15   121.3 1063.35     182 1046.48   212.3 1037.06   242.6 1022.95
   252.2  1019.4   271.4 1016.27   319.1 1004.16   329.1 1002.21   339.1 1002.68
   357.9 1006.51   367.5 1007.53   465.8  1014.7   475.9 1016.21     486 1019.53
   526.3 1039.07   556.5 1054.79   566.5 1058.58   576.6  1060.7   616.9 1084.32
   637.1 1097.69   677.3 1120.12   697.5 1128.96   707.6 1130.82   717.6 1136.16
#Mann= 3 , 0 , 0
       0     .06       0   319.1    .045       0   339.1     .06       0
Bank Sta=319.1,339.1
XS Rating Curve= 0 ,0
Exp/Cntr=0.3,0.1

Type RM Length L Ch R = 1 ,27982.2 ,360.2,349,337.8
XS GIS Cut Line= 4
     1644900.022      263617.578     1644947.212      263861.393
     1644951.931      264040.714     1645040.018      264306.551
#Sta/Elev= 30
     9.9 1101.51    19.9 1099.66    69.5 1076.53   119.2 1046.77   129.1 1046.32
   168.9 1023.78   188.7 1014.96   198.7 1011.92   218.5 1008.19   298.2 1003.16
   328.1  996.43     338  995.67     348  994.34     358  995.96   377.9 1000.91
   387.9 1004.33   437.7 1036.56   447.7 1037.31   537.7 1099.72   547.7 1104.04
   557.7 1106.98   587.8 1128.77   597.8 1134.12   627.8 1157.01   657.8 1177.04
   667.8 1179.65   677.8 1183.98   687.8 1190.06   697.8 1194.74   707.8  1198.1
#Mann= 3 , 0 , 0
       0     .06       0     338    .045       0     358     .06       0
Bank Sta=338,358
XS Rating Curve= 0 ,0
Exp/Cntr=0.3,0.1

Type RM Length L Ch R = 1 ,27633.2 ,285.7,279.4,273.1
XS GIS Cut Line= 4
     1644476.885      263829.933     1644580.703      263968.356
     1644656.207      264116.218      1644815.08      264338.011
#Sta/Elev= 30
     9.6 1124.15    48.1 1102.29    67.3 1090.44    86.5 1076.95    96.1 1075.29
   115.4 1063.86   192.6 1015.65   202.3 1008.83   212.1 1000.72   221.9  994.73
   231.4  992.81   241.4  989.02   251.4  990.99   260.9  994.67   270.7  995.93
   309.8  996.38   319.5  997.44   349.2 1005.06   359.3 1006.49   379.5  1012.5
   409.8 1025.64   440.1 1043.52   480.5 1063.73   490.6 1065.32   500.7 1069.09
     531 1083.44   551.2 1094.05   571.5 1106.33   581.6  1111.5   611.9 1130.68
#Mann= 3 , 0 , 0
       0     .06       0   231.4    .045       0   251.4     .06       0
Bank Sta=231.4,251.4
XS Rating Curve= 0 ,0
Exp/Cntr=0.3,0.1

Type RM Length L Ch R = 1 ,27353.9 ,302.1,303.4,304.8
XS GIS Cut Line= 4
     1644217.341      263991.951     1644335.316      264128.802
     1644429.696      264235.766     1644667.218       264421.38
#Sta/Elev= 30
      10 1117.28    20.1 1112.07    70.3  1091.7    80.3 1085.63   100.4  1071.2
   110.4 1066.51   120.5  1059.1   130.5 1056.11   150.6 1041.73   170.6 1024.38
   209.2  997.97   247.3   987.3   256.3  985.93   266.3  985.85   276.3  986.42
   304.3  990.28   373.6  995.67   383.6  997.94   393.7 1002.53   413.8 1017.78
   423.8 1023.39     454 1038.35     464 1041.09   494.2  1056.5   504.2 1062.51
   514.2 1070.06   594.6 1111.68   604.7  1117.4   614.7 1126.45   624.8 1133.01
#Mann= 3 , 0 , 0
       0     .08       0   256.3    .045       0   276.3     .08       0
Bank Sta=256.3,276.3
XS Rating Curve= 0 ,0
Exp/Cntr=0.3,0.1

Type RM Length L Ch R = 1 ,27050.4 ,344.6,352,359.3
XS GIS Cut Line= 4
     1644044.311      264108.353     1644149.702      264338.011
     1644258.239      264471.716     1644412.393       264715.53
#Sta/Elev= 30
    10.1 1101.66    40.4 1086.69    60.6 1081.35    80.9 1072.24      91 1067.29
   161.7 1023.98   171.8 1019.93   181.9 1018.58   202.1  1007.9   222.4   999.3
   252.7  993.52   343.9   983.4   364.2  978.97   374.2  978.54   384.2  981.75
   414.8  997.78   424.9 1004.07   434.8 1012.39   444.8 1018.07   454.7 1020.09
   464.7 1027.42   474.6 1032.46   514.4 1045.55   564.2 1060.31   574.1 1062.37
     584 1060.89   643.7 1076.31   673.6 1081.43   703.4  1089.9   713.4 1089.32
#Mann= 3 , 0 , 0
       0     .08       0   364.2    .045       0   384.2     .08       0
Bank Sta=364.2,384.2
XS Rating Curve= 0 ,0
Exp/Cntr=0.3,0.1

Type RM Length L Ch R = 1 ,26698.4 ,225.8,230.3,234.8
XS GIS Cut Line= 4
     1643736.004      264271.945     1643876.001      264496.884
     1643943.639      264662.048     1644105.658      264844.516
#Sta/Elev= 30
     9.8  1083.8    29.4 1070.87    58.9 1052.93    68.7  1051.7    78.5 1047.04
   147.2  999.62     157  994.05   166.8  990.12   186.4  986.12   196.3  984.93
   255.1  981.83   314.5  977.81   334.4  977.07  360.15  973.95     374  972.91
  379.94  975.09   383.9  976.67   393.8  984.54   403.8  991.09   433.5 1008.28
   443.4 1011.38   453.2 1013.64   531.3 1057.35     541 1064.01   580.1 1086.29
   589.8 1090.04   599.6 1091.06   638.6  1111.8   667.9 1123.25   687.4  1132.2
#Mann= 3 , 0 , 0
     9.8     .06       0  360.15    .045       0  379.94     .06       0
Bank Sta=360.15,379.94
XS Rating Curve= 0 ,0
Exp/Cntr=0.3,0.1

Type RM Length L Ch R = 1 ,26468.1 ,260.5,256.3,252
XS GIS Cut Line= 4
     1643579.611      264345.516      1643670.47      264544.269
     1643704.542      264704.691     1643825.213      264870.791
#Sta/Elev= 30
     9.9 1070.31    39.7 1052.16    69.5 1030.91    79.5 1026.64    89.4 1024.08
   129.1  998.22   139.1  993.96   198.7  982.84   208.6  982.51   237.8   978.2
   266.8  974.69   305.4  971.34     315  970.97   324.3  969.25   334.3  968.32
   344.3  971.03   363.2  982.32   372.9   986.6   382.5  990.38   402.1  996.78
   421.6 1005.41   431.4 1007.26   441.2 1009.88   490.1 1033.62   519.4 1048.78
   529.2 1054.18   548.7 1066.41   558.5 1070.72   578.1 1076.23   587.8 1080.49
#Mann= 3 , 0 , 0
       0     .06       0   324.3    .045       0   344.3     .06       0
Bank Sta=324.3,344.3
XS Rating Curve= 0 ,0
Exp/Cntr=0.3,0.1

Type RM Length L Ch R = 1 ,26211.8 ,223.1,210.7,198.3
XS GIS Cut Line= 4
     1643347.474      264396.212     1643391.517      264581.825
     1643463.875       264762.72     1643641.624      264934.177
#Sta/Elev= 30
      10    1089    20.1 1083.03    40.2 1068.98    90.4 1030.83   100.4 1029.64
   130.5 1009.87   140.6 1004.03   160.6  993.59   190.8  980.66   200.5  977.15
   210.3  975.29     220  974.67   249.2  968.92   297.9  967.42   326.9  964.31
   336.9  963.86   346.9  964.76   356.4  969.05   375.9  979.93   385.6  983.83
   395.5  987.66   415.2  992.51   425.1  995.92     435  998.03   484.4 1004.86
   523.9 1013.71   553.5 1025.68   602.9 1048.54   622.7 1056.69   632.6 1059.31
#Mann= 3 , 0 , 0
       0     .06       0   326.9    .045       0   346.9     .06       0
Bank Sta=326.9,346.9
XS Rating Curve= 0 ,0
Exp/Cntr=0.3,0.1

Type RM Length L Ch R = 1 ,26001.1 ,226.9,243.8,260.7
XS GIS Cut Line= 4
     1642923.726       264538.59     1643219.017      264796.969
     1643370.921      264924.739     1643527.084      265127.751
#Sta/Elev= 30
    10.1 1080.81    30.2 1076.91   110.7 1044.41   150.9 1031.07   181.1 1028.15
   191.2    1026   201.2 1020.94   211.3 1018.95   221.3 1015.36   251.5 1002.93
   321.9  977.43   362.2  970.09     442  963.43   461.8  959.31   471.8  958.18
   481.8  958.82   521.4  962.06   531.3  965.16   541.2  972.35   551.2  982.35
   561.1  986.54   600.7  992.94   610.6  996.15   689.4 1029.49   699.2 1035.19
   718.9    1043   728.8 1049.12   787.9 1079.34   837.1 1106.02     847 1109.01
#Mann= 3 , 0 , 0
       0     .06       0   461.8    .045       0   481.8     .06       0
Bank Sta=461.8,481.8
XS Rating Curve= 0 ,0
Exp/Cntr=0.3,0.1

Type RM Length L Ch R = 1 ,25757.4 ,189.5,193.5,197.5
XS GIS Cut Line= 4
     1642896.023      264536.209     1643054.896      264802.045
     1643105.232      265045.859     1643232.645      265266.079
#Sta/Elev= 30
      10 1082.87      20 1081.46      40 1073.32    89.9 1045.32   119.9 1030.23
   129.9 1026.01   139.9    1026   189.8 1004.59   259.7  977.19   269.7  977.25
   289.7  969.46   299.7  967.22   379.4  962.69   389.4  962.77   439.2   959.2
   488.9  954.88   498.9  954.04   508.9  954.39   518.8  959.08   538.7  974.13
   558.6   987.1   597.8 1011.19   617.4 1016.43   646.7 1034.87   666.3  1047.9
     725 1084.87   734.8  1088.5   744.6 1090.45   793.5 1119.53   813.1 1131.64
#Mann= 3 , 0 , 0
       0     .06       0   488.9    .045       0   508.9     .06       0
Bank Sta=488.9,508.9
XS Rating Curve= 0 ,0
Exp/Cntr=0.3,0.1

Type RM Length L Ch R = 1 ,25563.8 ,246.6,238.1,229.5
XS GIS Cut Line= 4
     1642757.626      264640.806     1642896.753      264900.604
     1642903.851      265061.026     1642962.057      265320.825
#Sta/Elev= 30
     9.8 1057.56    29.5  1044.2    58.9 1027.42   108.1 1001.36   117.9   998.9
   127.7  995.22     167  972.21   176.8  967.86   186.6  965.78   196.5  964.94
   284.9  961.11   344.9  955.56   354.9   955.5     375  952.59   385.1  949.88
   395.1  947.74   405.1  947.97   415.1  953.85   425.2  961.97   445.2  975.53
   455.3   976.6   465.1  981.94   553.9 1039.61   563.8 1044.33   573.6 1046.09
   632.8 1084.36   662.4 1104.19   672.2 1105.89   682.1 1110.26   721.5 1132.22
#Mann= 3 , 0 , 0
       0     .06       0   385.1    .045       0   405.1     .08       0
Bank Sta=385.1,405.1
XS Rating Curve= 0 ,0
Exp/Cntr=0.3,0.1

Type RM Length L Ch R = 1 ,25325.8 ,348.3,345.7,343.1
XS GIS Cut Line= 4
     1642507.493      264707.665     1642617.603      264931.031
     1642697.826      265127.655     1642903.888       265340.01
#Sta/Elev= 30
      10 1072.55    19.9 1066.84    39.8 1053.18    89.7 1021.89   109.6 1008.42
   129.5 1000.25   169.3  969.85   179.3   963.6   189.3  960.09   229.1  956.05
   319.8  948.72   370.4  946.93   380.6  945.44   390.6  944.35   400.6  945.85
   431.1  965.46   471.3  989.62   481.1  990.57     491  995.98   500.8  999.99
   540.3 1019.39   579.8 1039.95   609.3 1057.78   638.9 1073.53   648.8 1075.14
   658.7 1078.68   698.1 1100.39   717.8  1113.9   727.7 1118.75   757.3 1130.44
#Mann= 3 , 0 , 0
       0     .06       0   380.6    .045       0   400.6     .08       0
Bank Sta=380.6,400.6
XS Rating Curve= 0 ,0
Exp/Cntr=0.3,0.1

Type RM Length L Ch R = 1 ,24980.1 ,223.6,208.9,194.2
XS GIS Cut Line= 4
      1642276.36      264767.156     1642306.173      265110.715
     1642394.192      265275.396        1642698.      265448.595
#Sta/Elev= 30
     9.9 1074.91    19.7  1074.1    29.6 1069.66   108.4  1012.2   128.1 1005.58
   187.2  965.73   197.1  959.89   206.9  957.24   226.6  955.66   325.1  948.52
   423.5  942.91   433.3  942.01   452.8  938.12   462.8  937.81   472.8   938.4
   482.4  942.92   502.1   955.7   531.6  972.89   551.6  982.38   561.6   985.9
   601.5  988.69   641.5  996.09   661.5 1003.41   731.4 1020.61   751.4 1027.22
   781.4 1032.62   821.3 1041.92   831.3 1044.77   841.3 1050.65   881.3  1062.4
#Mann= 3 , 0 , 0
       0     .06       0   452.8    .045       0   472.8     .08       0
Bank Sta=452.8,472.8
XS Rating Curve= 0 ,0
Exp/Cntr=0.3,0.1

Type RM Length L Ch R = 1 ,24771.2 ,65.2,60.8,56.5
XS GIS Cut Line= 4
     1641859.418      265141.812     1642060.762      265273.944
     1642347.047      265428.098     1642560.975      265695.507
#Sta/Elev= 30
      10 1079.69    20.1 1073.69    30.1 1063.48   110.4 1015.99   130.4    1001
   180.6  976.33   210.7  963.51   220.8  957.58   240.8  952.11   368.9  938.91
   398.3  933.68   408.3  932.85   418.3  934.25   437.9  940.97   457.6  944.99
   546.3  953.45     566  953.48   576.1  955.85   586.1  960.41   596.2  970.13
   606.3  976.37   626.4  986.65     707 1013.17   717.1 1018.39   737.2 1034.82
   757.3 1044.55   837.9 1069.95   868.1 1080.15   878.2 1086.34   908.4 1095.18
#Mann= 3 , 0 , 0
       0     .06       0   398.3    .045       0   418.3     .06       0
Bank Sta=398.3,418.3
XS Rating Curve= 0 ,0
Exp/Cntr=0.3,0.1

Type RM Length L Ch R = 1 ,24710.3 ,215.1,209.4,203.8
XS GIS Cut Line= 4
     1641727.264      265326.409     1642089.057      265376.113
     1642252.038       265430.44     1642541.837      265697.036
#Sta/Elev= 30
     9.9 1131.56    29.6 1115.57    88.8 1085.63    98.7 1079.61   108.6 1070.82
   167.8 1040.92   177.7 1030.63   246.8  991.02   256.6  980.34   266.5  971.91
   325.7  937.87   335.6  935.67   425.8  936.12   446.1  933.17   456.1  931.42
   466.1  931.59   486.5  938.27   506.7  942.18   577.4  944.06   607.7  947.96
   617.8  950.88   648.1  965.54   698.5   981.5   708.6  987.86   759.1 1013.04
   809.6 1033.64   819.7 1040.75   910.6 1073.94   920.7 1078.71   930.8 1086.34
#Mann= 3 , 0 , 0
       0     .06       0   446.1    .045       0   466.1     .06       0
Bank Sta=446.1,466.1
XS Rating Curve= 0 ,0
Exp/Cntr=0.3,0.1

Type RM Length L Ch R = 1 ,24500.9 ,360,362.7,365.4
XS GIS Cut Line= 4
      1641676.95      265464.277     1641978.966      265593.263
     1642244.803      265618.431     1642538.953      265709.664
#Sta/Elev= 30
      10 1171.27    19.9 1162.71    89.6 1125.86   109.5 1108.72   179.1 1072.57
   189.1 1063.63     199 1057.59   268.7 1021.55   278.6  1010.7   338.3  975.13
   348.2  966.52   358.1  955.93   387.7  937.67   397.6  934.27   447.1  930.78
   466.8  926.34   476.8  925.24   486.8  925.49   516.3  931.31   625.2  940.35
   645.1  943.28     655  947.67     665  955.67   734.5  987.95   754.4 1002.24
   804.1 1026.39     814 1032.51   823.9  1041.3   893.5 1075.28   903.4 1083.72
#Mann= 3 , 0 , 0
       0     .06       0   466.8    .045       0   486.8     .06       0
Bank Sta=466.8,486.8
XS Rating Curve= 0 ,0
Exp/Cntr=0.3,0.1

Type RM Length L Ch R = 1 ,24138.2 ,442.3,447.8,453.2
XS GIS Cut Line= 4
     1641547.965      265967.636     1641953.798      265940.895
     1642229.072      265997.523     1642502.774      266109.205
#Sta/Elev= 30
     9.9 1115.63    39.7 1102.51    49.6 1094.81   109.1 1067.31     129 1055.53
   158.7 1043.75   178.6 1037.79   198.4 1028.93   257.9 1010.97   277.8 1002.52
   347.2  980.45     377  980.58   406.7  974.63   446.9  943.01   466.9  929.54
   507.1  919.72   517.1  918.72   527.1  919.17   607.5  929.47   637.6  939.47
   657.6  950.72   717.3  976.33   746.9  994.19     806 1022.39   815.8 1031.23
   825.7 1037.25   894.7 1072.48   904.5 1081.93   914.4 1087.32   983.4 1116.01
#Mann= 3 , 0 , 0
       0     .06       0   507.1    .045       0   527.1     .06       0
Bank Sta=507.1,527.1
XS Rating Curve= 0 ,0
Exp/Cntr=0.3,0.1

Type RM Length L Ch R = 1 ,23690.4 ,493.3,495.4,497.5
XS GIS Cut Line= 4
     1641513.359      266107.633     1641750.881      266307.403
     1642071.773      266450.546     1642280.981       266667.62
#Sta/Elev= 30
      10 1082.91      20 1076.89      40 1060.33    60.1 1048.06    80.1 1040.21
   120.1 1015.56   140.2  999.07   240.3  940.42   260.3  930.78   320.4  924.22
   370.6  924.13     471  917.93   491.1  914.29   501.1   912.6   511.1  916.78
   531.2  928.25   541.3  938.08   571.4   956.9   591.5  973.93   601.5  985.12
   611.5  991.64   671.8 1024.94   701.9 1046.26   762.2 1083.63   772.3 1085.57
   782.3 1090.56   852.7 1132.18     913 1172.41   933.1 1179.36   963.2 1199.24
#Mann= 3 , 0 , 0
       0     .06       0   491.1    .045       0   511.1     .06       0
Bank Sta=491.1,511.1
XS Rating Curve= 0 ,0
Exp/Cntr=0.3,0.1

Type RM Length L Ch R = 1 ,23195   ,194,202,210.1
XS GIS Cut Line= 4
      1641367.07      266533.915     1641558.976      266747.842
     1641736.724      266845.368     1641950.652      266884.693
#Sta/Elev= 30
     9.9  997.23    89.2  962.42    99.1  956.21     109  951.01   158.6  935.89
   178.4  931.79   188.3  928.92   198.2  925.46     218  916.82   227.9  913.98
   287.4  911.61   374.3  909.48   383.9  909.07  399.65     907   412.9  905.75
   417.8  908.45   422.6  911.31   432.2  919.42   441.9  926.35   461.2  938.65
   480.5  945.59     500   957.3   519.8  976.62   539.6  989.09   579.1  1009.2
     589 1017.52   658.2 1048.66   668.1 1056.81     678 1062.56   707.6  1077.3
#Mann= 3 , 0 , 0
     9.9     .06       0  399.65    .045       0   417.8     .06       0
Bank Sta=399.65,417.8
XS Rating Curve= 0 ,0
Exp/Cntr=0.3,0.1

Type RM Length L Ch R = 1 ,22993   ,373.2,373.2,373.3
XS GIS Cut Line= 4
     1641177.539       266652.47     1641417.463      266831.348
     1641575.046      267000.288     1641717.012      267105.343
#Sta/Elev= 30
      10  1045.5    29.9 1034.85    39.9 1028.33    49.9 1022.89    59.9 1015.91
   129.7   978.7   139.7  972.54   149.6  969.69   209.5  935.78   229.4  923.86
   239.4  917.11   249.4  911.74   259.4  910.04   269.3  909.73   439.9  907.14
   449.9  906.69   470.1  903.41   480.1   902.7   490.1  904.98   500.2  907.29
   549.9  941.35   559.7  948.36   579.4  963.67     599  981.15   608.8  984.35
   638.2  991.47     648  994.92   677.5 1010.82   687.3 1014.85   706.9 1027.55
#Mann= 3 , 0 , 0
       0     .06       0   470.1    .045       0   490.1     .06       0
Bank Sta=470.1,490.1
XS Rating Curve= 0 ,0
Exp/Cntr=0.3,0.1

Type RM Length L Ch R = 1 ,22619.8 ,214.8,213.5,212.1
XS GIS Cut Line= 4
     1641006.854      266716.382     1641115.391      267053.004
     1641299.431      267251.202     1641463.023      267342.435
#Sta/Elev= 30
    10.1 1089.67    30.3 1072.36    50.5 1056.13    70.7 1042.28    90.9  1030.3
   101.1 1027.84   111.2 1023.95   212.2  968.52   222.3  967.56   272.8     941
   313.3  917.35   333.5  911.96   343.6   907.7   353.7  905.39     514  900.96
     534  899.67     544  898.27     554     897     564  897.44   574.1  903.27
   584.1  918.78   594.1  931.57   624.2  961.35   643.9  968.58   673.4  986.26
   693.2  999.93   762.2 1033.75     772  1038.8   781.9 1045.54   811.5 1059.81
#Mann= 3 , 0 , 0
       0     .06       0     544    .045       0     564     .06       0
Bank Sta=544,564
XS Rating Curve= 0 ,0
Exp/Cntr=0.3,0.1

Type RM Length L Ch R = 1 ,22406.3 ,283,282.5,282
XS GIS Cut Line= 4
     1640770.096      266987.511     1641002.921      267252.988
     1641122.172      267367.981     1641434.499      267502.849
#Sta/Elev= 30
    10.1 1004.02    20.2  999.85    40.4  988.15    60.5  974.59     111  950.19
   141.2  939.37   151.3  936.54   161.4  936.01   171.5  932.72   242.1  905.91
   272.4  902.23   421.3  896.78   450.3  893.55   460.3  892.67   470.3  893.64
   479.8   895.6   489.5  902.96     509  922.93   528.8  940.55   538.8  951.89
   548.8  960.42   608.8  998.41   618.8 1008.06   658.9 1029.26   728.9 1062.34
   758.9 1080.47   788.9 1095.45   798.9 1103.53   808.9 1109.13     859 1135.02
#Mann= 3 , 0 , 0
       0     .06       0   450.3    .045       0   470.3     .06       0
Bank Sta=450.3,470.3
XS Rating Curve= 0 ,0
Exp/Cntr=0.3,0.1

Type RM Length L Ch R = 1 ,22123.8 ,491.9,501.5,511.1
XS GIS Cut Line= 4
     1640534.955      267101.767     1640747.309      267403.782
     1640954.945      267595.688     1641585.717      267691.641
#Sta/Elev= 30
      10 1042.72    79.8  996.76    99.8  987.48   149.7  954.55   219.5   915.4
   239.5   909.3   259.4  898.15   269.4   896.2   369.2  897.72     541  888.19
     551  887.39     561   887.7   571.2  894.14   611.5  940.89   641.8  964.18
   712.7  998.16   773.5 1021.56   793.7 1034.82   844.4 1058.57   864.6 1073.31
   874.7 1077.37   905.1 1086.39     976 1098.65  1006.4 1106.83  1016.5  1112.5
  1097.5 1130.63  1158.3 1139.91  1229.2 1164.08  1259.6 1169.78    1290 1170.09
#Mann= 3 , 0 , 0
       0     .06       0     541    .045       0     561     .06       0
Bank Sta=541,561
XS Rating Curve= 0 ,0
Exp/Cntr=0.3,0.1

Type RM Length L Ch R = 1 ,21622.3 ,458.2,455.4,452.6
XS GIS Cut Line= 4
     1639959.238      267510.746     1640470.021      267757.258
     1640593.058      268016.583     1640767.204      268345.946
#Sta/Elev= 30
    10.1 1021.28    70.9  992.87      81  985.66    91.2  975.76   151.9  940.45
     162  932.56   172.2   926.4   243.1  904.86   263.3  892.47   273.5  889.55
   293.7   887.6   526.6  888.35   606.7  887.34     676  884.04   695.7  879.23
   705.7  879.02   715.7  879.97     775  886.16   924.7  892.59   954.9  899.39
     965  899.91   995.2  913.12  1035.4  934.22  1075.7  952.45  1095.9   955.3
  1166.3  981.61  1196.5  994.14  1206.6  997.27  1216.7  996.38  1226.8 1000.55
#Mann= 3 , 0 , 0
       0     .06       0   695.7    .045       0   715.7     .06       0
Bank Sta=695.7,715.7
XS Rating Curve= 0 ,0
Exp/Cntr=0.3,0.1

Type RM Length L Ch R = 1 ,21166.9 ,158.5,172.3,186.2
XS GIS Cut Line= 4
     1639866.409      267631.219     1640011.623      267907.947
     1640217.115      268239.474     1640400.687      268538.121
#Sta/Elev= 30
    10.1 1035.37    40.3  1015.6    90.7  979.53   100.8  974.15   110.9  972.66
   211.7  902.68   221.8  901.04   241.9  890.33     252  888.05   262.1   887.5
   472.5  882.06   542.5  878.48   562.5  876.42   572.5  875.83   582.5  876.07
   592.5  878.77   602.6  886.03   612.6  888.78   652.6  909.77   732.6  948.15
   742.6  948.85   762.7  957.44   862.8 1016.15   872.8 1017.61   882.8 1021.72
   922.9 1044.85     993 1087.68    1003 1089.39  1013.1 1093.35  1053.1 1117.72
#Mann= 3 , 0 , 0
       0     .06       0   562.5    .045       0   582.5     .06       0
Bank Sta=562.5,582.5
XS Rating Curve= 0 ,0
Exp/Cntr=0.3,0.1

Type RM Length L Ch R = 1 ,20994.5 ,783.6,764,744.4
XS GIS Cut Line= 4
     1639830.252      267620.856     1639978.114      267971.634
     1639979.686      268267.358     1640050.471      268434.095
#Sta/Elev= 30
      10 1046.64    90.2  993.37   110.2  986.63   170.3  945.17   190.3  930.23
   210.4  917.13   220.4  912.42   230.4  909.14   250.4   895.4   260.5  890.06
   270.5  888.06   300.5   885.8   528.5  881.66   558.1  880.35   577.7  877.51
   587.7  875.82   597.7  877.66   607.4   887.2   617.3   902.4   627.1  910.78
   646.8  916.81   656.7  917.53   696.5  928.86   706.6  932.63   736.8   947.1
   756.9  959.48     777  966.06   807.2  984.07   817.3  988.49   857.5 1001.61
#Mann= 3 , 0 , 0
      10     .06       0   577.7    .045       0   597.7     .06       0
Bank Sta=577.7,597.7
XS Rating Curve= 0 ,0
Exp/Cntr=0.3,0.1

Type RM Length L Ch R = 1 ,20230.5 ,566,560.2,554.5
XS GIS Cut Line= 4
     1639128.695      267965.342     1639315.882      268113.204
     1639504.641      268301.964     1639660.368       268504.88
#Sta/Elev= 30
     9.9  1064.9    59.6 1033.41    69.6 1026.27    79.5 1020.13   139.1  992.04
     159   986.9     169  980.42   178.9  972.75   268.2   919.4     288  905.58
   307.7  895.23   317.6  891.91   327.5  886.35   337.4  883.87   357.1  871.73
   367.1  869.47   377.1   869.5   505.5  880.87     535   886.9   564.5  889.66
   574.4  892.55   603.9  903.02   613.7  905.68   623.5  905.89   633.4  907.85
   653.1   908.7   692.4  928.03   721.9  946.51   731.8  951.37   761.3   963.9
#Mann= 3 , 0 , 0
       0     .06       0   357.1    .045       0   377.1     .06       0
Bank Sta=357.1,377.1
XS Rating Curve= 0 ,0
Exp/Cntr=0.3,0.1

Type RM Length L Ch R = 1 ,19670.3 ,781.4,814.5,847.5
XS GIS Cut Line= 4
     1638641.066      268300.391     1638955.665      268534.767
     1639158.582      268673.191     1639342.623      268844.648
#Sta/Elev= 30
    10.1  1099.1    50.3 1079.96    60.4 1069.85   100.6 1049.71   150.9 1028.35
   160.9 1022.32   191.1 1009.08   211.2  1004.7   231.4  996.51   281.7  972.31
   352.1   941.7   362.1  932.95   382.2  919.69   402.1  909.01   421.8  901.42
   451.3  884.95   461.1  871.46   470.7  864.86   480.7  864.01   490.7  865.27
   510.2  869.11   678.2   877.7   718.4  884.21   748.6  885.62   758.7  890.01
   768.7  897.77   798.9  914.51     819   922.2   879.4  954.34   889.5  960.85
#Mann= 3 , 0 , 0
       0     .08       0   470.7    .045       0   490.7     .06       0
Bank Sta=470.7,490.7
XS Rating Curve= 0 ,0
Exp/Cntr=0.3,0.1

Type RM Length L Ch R = 1 ,18855.8 ,687,641.6,596.2
XS GIS Cut Line= 4
     1638593.876      268682.629     1638589.157      268984.644
     1638545.113      269108.911     1638677.245      269329.131
#Sta/Elev= 30
    10.1  927.18    20.1  923.52    30.2  923.02   100.7  892.37   120.8  884.22
   130.9  884.02     151  877.13   221.5  869.58   231.6  869.56   271.8  867.33
   339.7     867   349.1  866.19   358.6     864   367.4  860.94   377.4  859.16
   387.4  859.69   405.6  863.45   415.1  867.45   433.9  882.42   443.8  880.14
   483.3  903.31   522.8  928.11   542.5  939.57   562.3  949.97   572.2   950.9
   582.1  955.65   601.8  965.94   611.7  971.92   621.6  978.54   690.7 1012.16
#Mann= 3 , 0 , 0
       0     .06       0   367.4    .045       0   387.4     .06       0
Bank Sta=367.4,387.4
XS Rating Curve= 0 ,0
Exp/Cntr=0.3,0.1

Type RM Length L Ch R = 1 ,18214.2 ,393.4,407.3,421.1
XS GIS Cut Line= 4
     1637920.633      269138.798     1638125.123      269256.773
     1638348.489      269294.525     1638538.821      269377.894
#Sta/Elev= 30
     9.8  988.32    19.7  982.35    29.5  977.59    39.3  973.67    49.2  966.26
     118  930.18   127.9  922.29   137.7  917.48   167.2  904.51   206.6  888.59
   226.2  877.85   245.9  871.14   275.5  862.21     295   855.1     305  852.37
     315  852.61   334.6  855.21   364.1  856.81   383.8  859.98   403.5  861.54
   462.6  864.25   502.2  864.91   512.1  866.17     522  869.42   531.9  874.02
   541.8  880.68   551.7  888.51     611  919.61   630.8  934.97   670.4  956.26
#Mann= 3 , 0 , 0
       0     .08       0     295    .045       0     315     .06       0
Bank Sta=295,315
XS Rating Curve= 0 ,0
Exp/Cntr=0.3,0.1
